--- Var.prj (project) ---

Proj Title=Var
Current Plan=p02
Default Exp/Contr=0.3,0.1
SI Units
Geom File=g01
Geom File=g02
Flow File=f02
Plan File=p02
Y Axis Title=Elevation
X Axis Title(PF)=Main Channel Distance
X Axis Title(XS)=Station
BEGIN DESCRIPTION:
END DESCRIPTION:
DSS File=dss
DSS Export Rating Curves= 0
DSS Export Rating Curve Sorted= 0
DSS Export Volume Flow Curves= 0
DXF OffsetX= 0
DXF OffsetY= 0
DXF ScaleX= 1
DXF ScaleY= 10

--- Var.p02 (plan) ---

Plan Title=Var_Plan_steady
Program Version=5.01
Short Identifier=steady
Geom File=g01
Flow File=f02
Mixed Flow
K Sum by GR= 0
Std Step Tol= 0.003
Critical Tol= 0.003
Num of Std Step Trials= 20
Max Error Tol= 0.1
Flow Tol Ratio= 0.001
Split Flow NTrial= 30
Split Flow Tol= 0.006
Split Flow Ratio= 0.02
Log Output Level= 0
Friction Slope Method= 1
Unsteady Friction Slope Method= 2
Unsteady Bridges Friction Slope Method= 1
Parabolic Critical Depth
Global Vel Dist= 0 , 0 , 0
Global Log Level= 0
CheckData=True
Encroach Param=-1 ,0,0, 0
BEGIN DESCRIPTION:
This model uses a steady 300 m³/s US BC and a Rating curve for the DS BC to create steady flow conditions in the river.
END DESCRIPTION:
Computation Interval=1MIN
Output Interval=1HOUR
Instantaneous Interval=1HOUR
Mapping Interval=1HOUR
Run HTab= 0
Run UNet= 0
Run Sediment= 0
Run PostProcess= 0
Run WQNet= 0
Run RASMapper= 0
UNET Theta= 1
UNET Theta Warmup= 1
UNET ZTol= 0.006
UNET ZSATol= 0.006
UNET MxIter= 20
UNET Max Iter WO Improvement= 0
UNET MaxInSteps= 0
UNET DtIC= 0
UNET DtMin= 0
UNET MaxCRTS= 20
UNET WFStab= 2
UNET SFStab= 1
UNET WFX= 1
UNET SFX= 1
UNET DSS MLevel= 4
UNET Pardiso=0
UNET DZMax Abort= 30
UNET Use Existing IB Tables=-1
UNET Froude Reduction=False
UNET Froude Limit= 0.8
UNET Froude Power= 4
UNET Time Slicing=0,0, 5
UNET Junction Losses=0
UNET D1 Cores= 0
UNET D2 Coriolis=0
UNET D2 Cores= 0
UNET D2 Theta= 1
UNET D2 Theta Warmup= 1
UNET D2 Z Tol= 0.003
UNET D2 Volume Tol= 0.003
UNET D2 Max Iterations= 20
UNET D2 Equation= 0
UNET D2 RampUpFraction=0.1
UNET D2 TimeSlices= 1
UNET D2 BCVolumeCheck=0
UNET D1D2 MaxIter= 0
UNET D1D2 ZTol=0.003
UNET D1D2 QTol=0.1
UNET D1D2 MinQTol=0.03
DSS File=dss
Write IC File= 0
Write IC File at Fixed DateTime=0
Write IC File at Sim End=0
Echo Input=False
Echo Parameters=False
Echo Output=False
Write Detailed= 0
HDF Write Warmup=0
HDF Write Time Slices=0
HDF Flush=0
HDF Face Node Velocities=0
HDF Compression= 1
HDF Chunk Size= 1
HDF Spatial Parts= 1
HDF Use Max Rows=0
HDF Fixed Rows= 1
Calibration Method= 0
Calibration Iterations= 20
Calibration Max Change=0.05
Calibration Tolerance=0.2
Calibration Maximum=1.5
Calibration Minimum=0.5
Calibration Optimization Method= 1
WQ AD Non Conservative
WQ ULTIMATE=-1
WQ Max Comp Step=1HOUR
WQ Output Interval=15MIN
WQ Output Selected Increments= 0
WQ Output face flow=0
WQ Output face velocity=0
WQ Output face area=0
WQ Output face dispersion=0
WQ Output cell volume=0
WQ Output cell surface area=0
WQ Output cell continuity=0
WQ Output cumulative cell continuity=0
WQ Output face conc=0
WQ Output face dconc_dx=0
WQ Output face courant=0
WQ Output face peclet=0
WQ Output face adv mass=0
WQ Output face disp mass=0
WQ Output cell mass=0
WQ Output cell source sink temp=0
WQ Output nsm pathways=0
WQ Output nsm derived pathways=0
WQ Output MaxMinRange=-1
WQ Daily Max Min Mean=-1
WQ Daily Range=0
WQ Daily Time=0
WQ Create Restart=0
WQ Fixed Restart=0
WQ System Summary=0
WQ Write To DSS=0
WQ Use Fixed Temperature=0
Sorting and Armoring Iterations= 10
XS Update Threshold= 0.02
Bed Roughness Predictor= 0
Hydraulics Update Threshold= 0.02
Energy Slope Method= 1
Volume Change Method= 1
Sediment Retention Method= 0
XS Weighting Method= 0
Number of US Weighted Cross Sections= 1
Number of DS Weighted Cross Sections= 1
Upstream XS Weight=0
Main XS Weight=1
Downstream XS Weight=0
Number of DS XS's Weighted with US Boundary= 1
Upstream Boundary Weight= 1
Weight of XSs Associated with US Boundary= 0
Number of US XS's Weighted with DS Boundary= 1
Downstream Boundary Weight= 0.5
Weight of XSs Associated with DS Boundary= 0.5
Percentile Method= 0
Sediment Output Level= 4
Mass or Volume Output= 0
Output Increment Type= 1
Profile and TS Output Increment= 1
XS Output Flag= 0
XS Output Increment= 10
Write Gradation File= 0
Read Gradation Hotstart= 0
Write HDF5 File= 1
Write DSS Sediment File= 0
SV Curve= 0
Specific Gage Flag= 0

--- Var.p01 (plan) ---

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Plan Title=Var_Plan
Program Version=5.04
Short Identifier=1
Geom File=g01
Flow File=f01
Subcritical Flow
steady flow upstream 300, downstream normal depth
Computation Time Step Use Courant=        0
Computation Time Step Use Time Series=    0
Computation Time Step Count To Double=0
Computation Time Step Max Doubling=0
Computation Time Step Max Halving=0
Computation Time Step Residence Courant=0
UNET 1D Methodology=Finite Difference
Write Binary Output= 1

--- Var.f02 (steady flow) ---

Flow Title=Var_steady
Program Version=5.01
Number of Profiles= 1
Profile Names=PF 1
River Rch & RM=Var,Reach 1         ,24130.8
     300
Boundary for River Rch & Prof#=Var,Reach 1         , 1
Up Type= 3
Up Slope=0.03
Dn Type= 4
Dn Rating Curve # Pts= 41
       0-2.00985     300-.333146304.9336-.116738305.3609-.115824413.3696.0658368
  516.93.2106168638.3517.3691128     738.4888992854.8859.6214872954.8874.7260336
1062.406.83789521173.441.9390888 1273.441.0290051383.774 1.127151484.2261.209142
1584.2251.2911331685.5881.3740381792.752 1.455421892.752 1.531011992.7521.606296
2099.778 1.684632199.7791.7544292299.7781.8245332399.7781.8946372505.684 1.96596
2605.6852.0314922705.6852.0970242805.6842.1625562910.7312.2290023010.7322.290877
 3110.732.3524463210.7282.414016 3315.072.4777193415.0992.5359363515.0982.594458
3615.0982.6526743715.0992.7108913818.9262.7697183918.9272.8251913999.7242.869997
4000.0012.870301
DSS Import GetInterval= 0
DSS Import GetPeak= 0
DSS Import FillOption= 0

--- Var.f01 (steady flow) ---

Flow Title=Var_Flow
Program Version=5.01
Number of Profiles= 1
Profile Names=PF 1
River Rch & RM=Var,1               ,24012.50
     300
Boundary for River Rch & Prof#=Var,1               , 1
Up Type= 3
Up Slope=0.001
Dn Type= 3
Dn Slope=0.001
DSS Import GetInterval= 0
DSS Import GetPeak= 0
DSS Import FillOption= 0

--- Var.g01 (geometry) ---

Geom Title=Var_Geometry
Program Version=5.01

River Reach=Var             ,Reach 1
Reach XY= 30
         990450.         184280.         990530.         183620.
         990130.         181460.         989980.         180820.
         989890.         180650.         989900.         180080.
         990110.         179450.         990280.         179230.
         990680.         178770.         991250.         178240.
         992280.         177080.         992360.         176960.
         992530.         176370.         992540.         176020.
         992470.         175650.         992352.         175342.
         991720.         174450.         990350.         172340.
         990190.         171940.         990070.         171270.
         990490.         168400.         990600.         167980.
         990690.         167100.         990960.         165690.
         991520.         164240.         991610.         164150.
         991750.         163620.         992050.         162900.
         992120.         162410.         992060.         162220.

Type RM Length L Ch R = 1 ,24130.8 ,9.939,9.939,9.939
BEGIN DESCRIPTION:
Topo1  0.000
END DESCRIPTION:
XS GIS Cut Line= 3
990520.149784416 184292.37937372         990450.         184280.
990379.850215584 184267.62062628
#Sta/Elev= 28
       0 132.793   9.643 132.498  11.752 132.726   19.33 132.793  19.821 132.791
   21.09 132.748  23.542 131.582  25.656  131.66  30.182  128.84  40.444 128.569
  51.938 128.407  54.867 126.012  63.454 126.361  68.149 130.266  70.887 130.403
  74.199 130.569  78.411 127.422  90.649 127.221  94.071 129.171 100.207 129.486
 107.197 127.354 109.696 126.654 117.319 126.646 120.397 127.272 121.804 128.191
 136.203 128.172 140.924 129.539 142.467 137.658
#Mann= 3 , 0 , 0
       0    .033       0       0    .033       0 142.467    .033       0
Bank Sta=0,142.467
XS Rating Curve= 0 ,0
Exp/Cntr=0.3,0.1

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
Type RM Length L Ch R = 1 ,23464.92,9.869,9.869,9.869
BEGIN DESCRIPTION:
Topo1  665.878
END DESCRIPTION:
XS GIS Cut Line= 3
990645.059757475 183612.57509813990529.998852009183619.994068712
990414.937946543183627.413039293
#Sta/Elev= 29
       0 129.803   2.212 129.771   2.419 128.129  11.381 128.146  11.878 128.448
  14.006 128.553   22.95   128.3  26.691 126.209  27.969 126.186  33.097  122.92
  48.064 123.321  49.713 123.939  64.298 123.719  73.088 125.547  94.846 124.414
 112.882 124.292 130.655 123.715 134.892 122.075 138.892 121.075 174.688  121.61
 178.708 122.067 187.259 123.711 201.464 123.682 203.726 122.904 208.814  122.52
 210.081 122.042 219.074 122.575 225.758 128.268 230.599 128.122
#Mann= 3 , 0 , 0
       0    .033       0       0    .033       0 230.599    .033       0
Bank Sta=0,230.599
XS Rating Curve= 0 ,0
Exp/Cntr=0.3,0.1

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
Type RM Length L Ch R = 1 ,22853.03,9.945,9.945,9.945
BEGIN DESCRIPTION:
Topo1  1277.773
END DESCRIPTION:
XS GIS Cut Line= 3
990525.496182238182999.812708077990409.998596359 183019.99017451
990294.501010479183040.167640943
#Sta/Elev= 29
       0 127.532    .929 127.667   4.105 127.631   7.555 127.271  11.136 123.429
  15.146 122.985  17.378 119.671  24.326 120.965  36.123 120.874  38.334 122.012
  55.919  122.03  73.417 122.124   83.58 122.119  92.913 122.115 110.505 122.111
 121.143 122.206 134.194 121.331 139.141 120.632 141.141 119.332 171.248 120.966
 177.576  121.32 188.814 121.578  198.96 121.664 210.806 120.589 215.359 120.318
 221.074 120.559 223.251 121.427 230.721 125.164 234.493 129.814
#Mann= 3 , 0 , 0
       0    .033       0       0    .033       0 234.493    .033       0
Bank Sta=0,234.493
XS Rating Curve= 0 ,0
Exp/Cntr=0.3,0.1

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
Type RM Length L Ch R = 1 ,22236.42,9.855,9.855,9.855
BEGIN DESCRIPTION:
Topo1  1894.382
END DESCRIPTION:
XS GIS Cut Line= 3
990430.989509829182393.806013829990319.997659474182409.981509841
990209.005809119182426.157005854
#Sta/Elev= 30
       0 123.744    8.35 123.817  14.328 123.756  19.829 118.905  24.931 116.225
  29.415 116.319  31.258 117.346  44.163 117.485  45.793  118.01  53.704 117.637
   59.21 117.844  60.226 118.131  68.665 117.564  72.672 119.255  79.567 119.032
    82.4 120.717  86.932 118.686  105.31 117.173 112.264 118.101 131.252 118.168
 146.392 117.533 148.392 115.883 164.496 116.648 165.944 117.491 187.722  118.73
 195.684 118.901 200.366 119.873  201.87 119.182 216.957 123.318 224.328  123.71
#Mann= 3 , 0 , 0
       0    .033       0       0    .033       0 224.328    .033       0
Bank Sta=0,224.328
XS Rating Curve= 0 ,0
Exp/Cntr=0.3,0.1

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
Type RM Length L Ch R = 1 ,21566.3 ,9.808,9.808,9.808
BEGIN DESCRIPTION:
Topo1  2564.502
END DESCRIPTION:
XS GIS Cut Line= 3
990290.534399541 181747.31263537         990180.181759.975198479
990069.465600459181772.637761587
#Sta/Elev= 25
       0 119.178   3.809 119.178   6.029 118.991  18.256 110.309  32.576 109.967
  48.857 110.463  68.741 111.693  82.739 111.218  85.727 107.924  93.826 106.505
 103.249 106.432  105.97 105.282 114.024 105.578 133.967 105.448 146.871 106.231
 157.593 105.662 187.262 105.585 193.397 106.142 201.831  107.41 208.088 110.571
 209.567 112.898 214.129 115.719 217.531 118.994 219.309 118.938 222.514 118.994
#Mann= 3 , 0 , 0
       0    .033       0       0    .033       0 222.514    .033       0
Bank Sta=0,222.514
XS Rating Curve= 0 ,0
Exp/Cntr=0.3,0.1

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
Type RM Length L Ch R = 1 ,21281.88,9.977,9.977,9.977
BEGIN DESCRIPTION:
Topo1  2848.929
END DESCRIPTION:
XS GIS Cut Line= 3
990241.324150189181455.146472197990133.513283583181479.674388065
990025.702416977181504.202303934
#Sta/Elev= 23
       0  117.54   3.991  117.54   7.831 117.213   16.89 109.037  35.318 110.361
  46.187 108.406   69.38 108.511  83.702 108.953  93.004 107.138 115.183 106.556
 136.372 105.307 147.598 104.666  160.16 104.612 163.359     105 174.855 105.023
 187.427 104.897 198.865 104.801 204.225 105.442 209.738 111.567 211.055 111.544
 216.823 117.236  218.02 117.203 221.131 117.236
#Mann= 3 , 0 , 0
       0    .033       0       0    .033       0 221.131    .033       0
Bank Sta=0,221.131
XS Rating Curve= 0 ,0
Exp/Cntr=0.3,0.1

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
Type RM Length L Ch R = 1 ,20623.41,9.618,9.618,9.618
BEGIN DESCRIPTION:
Topo1  3507.392
END DESCRIPTION:
XS GIS Cut Line= 3
990092.958026981180805.390332246989983.470560554180839.666509806
989873.983094128180873.942687367
#Sta/Elev= 25
       0 112.719    4.24 112.719   6.689 112.306  14.785 105.224  24.869 104.546
  25.577 103.049  34.677 101.809  54.945 101.941  71.274 102.747  88.121 103.329
  106.37 103.584 124.631 103.645 142.987 103.581 161.508  103.58 172.261 103.161
 180.441 103.001 181.608 102.418 183.444 101.736 209.314   101.4 212.653 102.444
 218.034  107.71 220.806 107.966 225.618 112.801 226.065 112.807 229.454 112.852
#Mann= 3 , 0 , 0
       0    .033       0       0    .033       0 229.454    .033       0
Bank Sta=0,229.454
XS Rating Curve= 0 ,0
Exp/Cntr=0.3,0.1

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
Type RM Length L Ch R = 1 ,20431.06,9.78,9.78,9.78
BEGIN DESCRIPTION:
Topo1  3699.746
END DESCRIPTION:
XS GIS Cut Line= 3
990104.236209226180621.457384599989899.344960098180667.651591296
 989694.45371097180713.845797993
#Sta/Elev= 30
       0 111.737   3.486 111.882   6.802 111.228  17.711 103.235  21.874 101.396
  38.706 102.001  60.185 101.569 122.695 102.836 162.975 102.879 164.629 101.175
 166.178 100.415  183.37 100.468  192.68 101.203 207.484 101.773 224.175 101.954
 246.038 101.561 258.355 102.122 276.149  101.48 291.196 103.489 323.837 102.838
 343.832 103.149 346.727 101.976 367.679 102.526 382.713 102.241 384.239 101.431
 393.587 100.944 399.597 101.012 401.036 101.538 412.102 110.607 420.067 110.494
#Mann= 3 , 0 , 0
       0    .033       0       0    .033       0 420.067    .033       0
Bank Sta=0,420.067
XS Rating Curve= 0 ,0
Exp/Cntr=0.3,0.1

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
Type RM Length L Ch R = 1 ,20010.54,9.396,9.396,9.396
BEGIN DESCRIPTION:
Topo1  4120.264
END DESCRIPTION:
XS GIS Cut Line= 3
  990059.8763594180250.952423394989908.671382021180249.929269685
989757.466404642180248.906115976
#Sta/Elev= 23
       0 108.517     4.2 108.594  15.329 103.633  24.524 102.009  38.439  101.57
  41.588  99.981  55.011   99.13  67.841   99.67  80.107  99.978  93.142 100.302
 105.611 100.102 119.576 100.049 132.052 100.214 159.858   99.21 161.779  98.581
 163.306  98.344 234.432  96.898 259.916  97.227 274.025  97.348 281.868 101.522
 293.121 107.981  294.19 108.006 302.416 108.195
#Mann= 3 , 0 , 0
       0    .033       0       0    .033       0 302.416    .033       0
Bank Sta=0,302.416
XS Rating Curve= 0 ,0
Exp/Cntr=0.3,0.1

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
Type RM Length L Ch R = 1 ,19860.21,9.818,9.818,9.818
BEGIN DESCRIPTION:
Topo1  4270.597
END DESCRIPTION:
XS GIS Cut Line= 3
990046.819309857180118.629269499989901.328652514180099.929787717
989755.837995172180081.230305935
#Sta/Elev= 28
       0 107.536    3.93 107.536  12.641 105.166  19.287 100.877  43.305 100.506
  59.522 101.333  75.793 101.827   79.47  98.504  84.902  98.363  87.687  99.218
  97.684  99.369 109.202  98.947 124.336  98.772 139.156  98.927 152.364  98.815
 157.612  97.443 172.862  98.097  200.87  98.225 212.373  97.899   227.2  97.745
 233.463  96.648 241.375  97.059 266.864  95.019 276.728 101.503 281.153 105.357
 283.672 105.596 284.883 106.787 293.374   106.9
#Mann= 3 , 0 , 0
       0    .033       0       0    .033       0 293.374    .033       0
Bank Sta=0,293.374
XS Rating Curve= 0 ,0
Exp/Cntr=0.3,0.1

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
Type RM Length L Ch R = 1 ,19565.68,9.502,9.502,9.502
BEGIN DESCRIPTION:
Topo1  4565.122
END DESCRIPTION:
XS GIS Cut Line= 3
 990130.47200864179860.549713244989984.854275984179819.296465059
989839.236543328179778.043216874
#Sta/Elev= 26
       0  105.25    4.15  105.25   7.031 104.746  19.392  97.486  40.843  97.526
   63.28  98.115  75.881   97.97  82.402  95.844 103.182  96.508 124.379  96.833
 144.667  97.024 165.494  96.838 187.239  96.824 202.919  97.096 213.679  95.416
  233.25  96.087  245.52  95.621 256.414  94.982 264.412   94.98 273.218  94.027
 279.216  94.327 280.918  95.197 285.459  97.291 294.972 104.885  295.66 104.903
 302.696 105.085
#Mann= 3 , 0 , 0
       0    .033       0       0    .033       0 302.696    .033       0
Bank Sta=0,302.696
XS Rating Curve= 0 ,0
Exp/Cntr=0.3,0.1

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
Type RM Length L Ch R = 1 ,19451.66,9.865,9.865,9.865
BEGIN DESCRIPTION:
Topo1  4679.140
END DESCRIPTION:
XS GIS Cut Line= 3
990159.010883454179757.151272979990014.746338552 179709.26342531
 989870.48179365179661.375577641
#Sta/Elev= 27
       0 104.466   3.971 104.466   7.501  103.44  17.735   96.82  34.671   96.93
   53.71   97.09  73.441   97.03  75.026  95.759  88.752  96.125 109.651  96.558
 113.931  95.722 131.387  95.597 148.418  95.836 167.022  96.309  188.33  96.135
 191.437  95.287 202.122   95.13 216.322  95.169 232.358  96.068 256.089  94.824
 260.787  94.421 277.442  92.854 283.441  94.854 289.231  98.412 295.161  104.02
  296.14 104.017 304.009 103.992
#Mann= 3 , 0 , 0
       0    .033       0       0    .033       0 304.009    .033       0
Bank Sta=0,304.009
XS Rating Curve= 0 ,0
Exp/Cntr=0.3,0.1

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
Type RM Length L Ch R = 1 ,19195.17,9.762,9.762,9.762
BEGIN DESCRIPTION:
Topo1  4935.631
END DESCRIPTION:
XS GIS Cut Line= 3
990230.612115753 179536.91658747990103.685143988179468.944568036
989976.758172223179400.972548602
#Sta/Elev= 28
       0 102.517   3.834 102.517    6.09 102.071  16.926  95.036  30.992  95.373
  45.713  94.961  61.162  94.765  76.451  94.223   80.46  93.583  93.266  93.636
  98.172  94.527 112.722  94.792 129.627  94.888  145.97  94.753 174.964  94.593
 176.896  93.395 178.499  92.783 185.248   91.64 193.248   92.64 209.213  93.317
 228.441  94.024 246.462  94.215 258.807  93.881 273.078  93.362 273.729  93.799
 279.685  99.754 280.571  99.751 287.962  99.754
#Mann= 3 , 0 , 0
       0    .033       0       0    .033       0 287.962    .033       0
Bank Sta=0,287.962
XS Rating Curve= 0 ,0
Exp/Cntr=0.3,0.1

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
Type RM Length L Ch R = 1 ,19038.97,9.39,9.39,9.39
BEGIN DESCRIPTION:
Topo1  5091.836
END DESCRIPTION:
XS GIS Cut Line= 3
990302.241440382179426.697859952990197.213044206179345.344346952
990092.184648031179263.990833953
#Sta/Elev= 27
       0 101.534   4.014 101.534   6.041  101.15  16.303  92.234  31.274  92.443
  41.415  92.211  44.068  93.552  68.997  93.893  84.792  93.915  99.226  93.976
 113.982  94.006 128.192  93.931 143.127  93.867 160.661  93.543 169.965  92.753
 184.057   92.24 186.351  91.783 194.398  90.826 204.399  91.326 207.055  92.186
 222.484  93.395 235.224  92.826 237.614  91.867 251.374  91.941 257.778  98.628
 259.509  98.637 265.701  98.671
#Mann= 3 , 0 , 0
       0    .033       0       0    .033       0 265.701    .033       0
Bank Sta=0,265.701
XS Rating Curve= 0 ,0
Exp/Cntr=0.3,0.1

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
Type RM Length L Ch R = 1 ,18916.9 ,9.982,9.982,9.982
BEGIN DESCRIPTION:
Topo1  5213.902
END DESCRIPTION:
XS GIS Cut Line= 3
990367.219396419179328.298351946990268.548494132179246.359294097
990169.877591845179164.420236248
#Sta/Elev= 24
       0 100.619   3.903 100.619   6.059  100.22  18.481  90.851  26.833  90.954
  28.771  91.742  45.115  92.936  58.716  93.072  74.144  92.986  95.131  93.088
 115.502  93.053 135.452  92.956 156.017  92.722 177.248  92.193 195.284  92.264
 213.049  91.692 216.138  91.256 228.115   89.46 238.115   90.96 240.008  91.672
 243.414  93.591 248.915  97.727 249.397  97.721 256.514  97.727
#Mann= 3 , 0 , 0
       0    .033       0       0    .033       0 256.514    .033       0
Bank Sta=0,256.514
XS Rating Curve= 0 ,0
Exp/Cntr=0.3,0.1

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
Type RM Length L Ch R = 1 ,18747.2 ,9.89,9.89,9.89
BEGIN DESCRIPTION:
Topo1  5383.607
END DESCRIPTION:
XS GIS Cut Line= 3
990482.953604323179208.527222899990385.876112819179124.123887181
990288.798621316179039.720551462
#Sta/Elev= 22
       0  99.381   3.812  99.381   5.919  99.001    18.8   89.91  42.145   90.27
  57.925  91.493  78.414  92.104  98.146  92.253  116.83  92.329 136.777  92.467
 156.623  92.348 175.076  91.867 177.084  91.207 179.133   90.57 189.131   90.27
 226.011  90.368  236.01  90.768 241.088  91.314 245.434  92.993  249.36   96.63
 250.068  96.624 257.277   96.63
#Mann= 3 , 0 , 0
       0    .033       0       0    .033       0 257.277    .033       0
Bank Sta=0,257.277
XS Rating Curve= 0 ,0
Exp/Cntr=0.3,0.1

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
Type RM Length L Ch R = 1 ,18440.61,9.715,9.715,9.715
BEGIN DESCRIPTION:
Topo1  5690.190
END DESCRIPTION:
XS GIS Cut Line= 3
 990680.79447581178980.196574774990585.161593042178893.354566262
990489.528710274 178806.51255775
#Sta/Elev= 25
       0   96.98   3.924   96.98    6.06  96.506  14.549  89.347  29.795  89.218
  31.025  89.692  62.517   89.98  82.437   89.87 101.082  89.621 120.565  89.871
 141.279  90.423 142.273  89.842 152.801  89.682 171.843  90.137 191.504  90.386
 194.758  89.542 198.204  89.183 213.204  88.493 233.232  87.899 241.232  88.199
 243.234  89.074 245.694  89.787 251.012  94.542 252.712  94.512 258.357  94.542
#Mann= 3 , 0 , 0
       0    .033       0       0    .033       0 258.357    .033       0
Bank Sta=0,258.357
XS Rating Curve= 0 ,0
Exp/Cntr=0.3,0.1

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
Type RM Length L Ch R = 1 ,18304.6 ,9.892,9.892,9.892
BEGIN DESCRIPTION:
Topo1  5826.205
END DESCRIPTION:
XS GIS Cut Line= 3
990762.761749328178875.391789655990668.256368042178786.147493942
990573.750986756178696.903198229
#Sta/Elev= 24
       0  95.892   4.034  95.892   7.267  94.921  15.244    88.5  17.795  87.945
  32.025  88.559  34.486  89.043  55.382  89.394  74.308  89.342  93.469  89.184
 111.448  89.135 132.046   88.51 140.794  88.517 142.765  89.228  163.85  89.533
 194.449  89.575  199.45   88.88 206.622  88.338 233.329   87.39 243.329   87.89
 245.321  88.868 252.024  93.682 252.524  93.668 259.967  93.682
#Mann= 3 , 0 , 0
       0    .033       0       0    .033       0 259.967    .033       0
Bank Sta=0,259.967
XS Rating Curve= 0 ,0
Exp/Cntr=0.3,0.1

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
Type RM Length L Ch R = 1 ,18126.55,9.991,9.991,9.991
BEGIN DESCRIPTION:
Topo1  6004.250
END DESCRIPTION:
XS GIS Cut Line= 3
990891.697397259178768.691391282990804.305288119178672.331559335
990716.913178979178575.971727388
#Sta/Elev= 30
       0  94.857   3.942  94.857   7.099  94.355  14.974  87.942  26.535  88.026
   30.63  88.278  33.754  87.664  45.439  87.615  49.754  88.343   72.67  88.761
  92.021  88.533 101.332  87.644 116.842   87.64 130.963  88.157 150.552  88.321
 169.666  88.641  173.12  88.106 180.612  87.826 193.304  87.068 201.303  87.468
 207.721  88.097 207.731  88.098 221.403  88.606 235.928  88.094 239.754  87.138
 245.795  86.979 247.039   88.04 252.427  92.749 253.174  92.746 260.173  92.718
#Mann= 3 , 0 , 0
       0    .033       0       0    .033       0 260.173    .033       0
Bank Sta=0,260.173
XS Rating Curve= 0 ,0
Exp/Cntr=0.3,0.1

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
Type RM Length L Ch R = 1 ,17786.84,9.609,9.609,9.609
BEGIN DESCRIPTION:
Topo1  6343.960
END DESCRIPTION:
XS GIS Cut Line= 3
 991134.21701036178530.533837097991045.374051856178433.581237562
990956.531093352178336.628638027
#Sta/Elev= 28
       0  93.148   3.943  93.148    5.89   92.73  18.828  88.642  18.962  86.894
  20.787  86.128  33.348  86.205  54.567   86.96  72.895  87.227  94.223  87.145
 113.521  87.043 132.241  86.688 138.157  86.082 140.936  85.517 146.935  85.317
 156.912  85.542 166.912  85.542   176.1   86.07 196.144  85.876 214.428  85.621
   232.3   85.12 238.877  84.175 246.818  85.235 247.536  86.541 250.952  87.117
 255.449  90.928 256.354  90.934 263.004  90.981
#Mann= 3 , 0 , 0
       0    .033       0       0    .033       0 263.004    .033       0
Bank Sta=0,263.004
XS Rating Curve= 0 ,0
Exp/Cntr=0.3,0.1

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
Type RM Length L Ch R = 1 ,17652.31,9.849,9.849,9.849
BEGIN DESCRIPTION:
Topo1  6478.496
END DESCRIPTION:
XS GIS Cut Line= 3
991238.941474906178442.717765358 991145.15937764178343.356560124
991051.377280373178243.995354891
#Sta/Elev= 29
       0  92.194   3.583  92.194   6.129  91.846  13.172  87.789  33.199  87.238
  34.784  85.598  41.011   85.36  42.552  84.423  57.307  84.432  57.398  84.429
   58.27  84.709  77.492  84.901  96.984  85.097 115.929  85.507 134.892  85.444
 154.773  85.532  174.46   85.81 193.937  85.975 217.037  85.417 219.692  84.553
  221.82  84.109 241.267  83.002 251.268  83.502 253.316  84.515  256.15  86.828
 260.621  86.765 260.681  89.771 262.323  89.785 273.259  89.881
#Mann= 3 , 0 , 0
       0    .033       0       0    .033       0 273.259    .033       0
Bank Sta=0,273.259
XS Rating Curve= 0 ,0
Exp/Cntr=0.3,0.1

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
Type RM Length L Ch R = 1 ,17346.98,9.869,9.869,9.869
BEGIN DESCRIPTION:
Topo1  6783.821
END DESCRIPTION:
XS GIS Cut Line= 3
991451.212969188178205.957235633991347.670582433178115.691985994
991244.128195679178025.426736355
#Sta/Elev= 30
       0  90.277   3.824  90.277   8.331  89.715   8.582  87.039   9.492  86.633
  14.031  82.545  31.834  82.493  34.955  83.007  54.193  83.798  71.099  84.191
  89.143  83.188 101.597  83.156 114.462  83.166 117.027  82.466 125.407  82.537
 130.959   84.26 149.981   84.82 161.478  83.728 182.269  84.347  200.75  84.469
 219.347  84.311  221.17  83.444 222.995  83.048 247.183  82.737 258.183  82.737
 260.893  83.476 263.916  85.165 266.673  87.595  267.71  87.602 274.727  87.647
#Mann= 3 , 0 , 0
       0    .033       0       0    .033       0 274.727    .033       0
Bank Sta=0,274.727
XS Rating Curve= 0 ,0
Exp/Cntr=0.3,0.1

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
Type RM Length L Ch R = 1 ,16764.68,9.475,9.475,9.475
BEGIN DESCRIPTION:
Topo1  7366.122
END DESCRIPTION:
XS GIS Cut Line= 3
991851.213460953177786.675322629991746.575952725177694.766452002
991641.938444497177602.857581376
#Sta/Elev= 27
       0  85.941   3.952  85.941   6.918  85.613  14.304  80.791  36.915  80.805
   40.41  81.333  58.216  81.327   76.91  81.246  95.331  81.208 114.155   81.01
 132.685  80.606 153.359  80.245 154.666  79.692 159.653  79.835 173.648  80.574
 193.366  80.346 225.046  79.697 231.999  79.732 238.223  80.063 247.159  79.778
 253.448  79.072 263.855  79.154 264.479  79.819 267.617  81.166  270.34   83.47
  273.01  83.527  278.54  83.709
#Mann= 3 , 0 , 0
       0    .033       0       0    .033       0  278.54    .033       0
Bank Sta=0,278.54
XS Rating Curve= 0 ,0
Exp/Cntr=0.3,0.1

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
Type RM Length L Ch R = 1 ,16622.56,9.806,9.806,9.806
BEGIN DESCRIPTION:
Topo1  7508.249
END DESCRIPTION:
XS GIS Cut Line= 3
991945.293046077 177674.35560735991837.358318059177585.450944594
991729.423590042177496.546281839
#Sta/Elev= 28
       0   85.03   3.912   85.03   6.239  84.508  11.951  80.802  30.098  80.103
  44.399  80.137  54.152  79.919  72.417  80.485   90.73  80.344 108.563  80.228
 125.229  80.029 142.828  79.802 144.325  79.139 160.993   78.86 170.512  79.032
 174.159  79.498 192.557  79.854 211.724  80.094 221.451  79.992 222.592  79.657
 233.795  79.473  239.95  78.886 265.172  78.161 265.738  79.465 267.581  80.379
 271.095  82.747 272.783  82.739  279.67  82.981
#Mann= 3 , 0 , 0
       0    .033       0       0    .033       0  279.67    .033       0
Bank Sta=0,279.67
XS Rating Curve= 0 ,0
Exp/Cntr=0.3,0.1

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
Type RM Length L Ch R = 1 ,16142.05,9.674,9.674,9.674
BEGIN DESCRIPTION:
Topo1  7988.752
END DESCRIPTION:
XS GIS Cut Line= 3
992262.453052582177329.369139495992158.638119669177231.361880331
992054.823186756177133.354621168
#Sta/Elev= 30
       0  82.196   3.882  82.417    5.72  82.174   8.181  80.063  11.781  80.054
  15.945  77.201  23.454  77.372  28.247    74.6   37.14  75.027  45.902  73.242
  46.687  72.708  55.088  72.276  65.278  72.155  71.621  73.041   78.86  72.811
  83.147  73.257 101.614   73.94 116.656  74.091 129.889  73.785 147.491  72.889
 179.077  72.896 214.228  72.337 233.201   72.73 262.387  73.877  265.63  75.897
 269.956  76.879 273.425  79.184 277.873  79.561 278.111  79.883 285.537  79.794
#Mann= 3 , 0 , 0
       0    .033       0       0    .033       0 285.537    .033       0
Bank Sta=0,285.537
XS Rating Curve= 0 ,0
Exp/Cntr=0.3,0.1

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
Type RM Length L Ch R = 1 ,15967.91,9.678,9.678,9.678
BEGIN DESCRIPTION:
Topo1  8162.893
END DESCRIPTION:
XS GIS Cut Line= 3
992384.519776199177183.384787316992265.661339232177094.338660768
992146.802902264177005.292534221
#Sta/Elev= 28
       0      82   4.004      82    6.01  81.015  14.648  75.998  30.173   75.71
  31.335  76.435  36.867  71.997   38.24  71.576  49.523  72.376  55.406  71.997
   74.89  72.173  86.443  71.828 116.602  71.652 126.118  72.316 128.087  74.351
 140.865  74.662 160.444  74.921 197.374  74.796 214.922  74.348 231.041  74.482
 245.532  73.858 262.673  73.914 275.238  73.325 280.988  73.853 284.265   74.97
 288.399  78.801 291.111  80.028 297.028  80.442
#Mann= 3 , 0 , 0
       0    .033       0       0    .033       0 297.028    .033       0
Bank Sta=0,297.028
XS Rating Curve= 0 ,0
Exp/Cntr=0.3,0.1

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
Type RM Length L Ch R = 1 ,15667.89,9.878,9.878,9.878
BEGIN DESCRIPTION:
Topo1  8462.918
END DESCRIPTION:
XS GIS Cut Line= 3
992540.439483719176881.132349678992397.986150406176830.034623984
992255.532817094176778.936898291
#Sta/Elev= 30
       0  79.436   4.853  79.436   7.519  79.074  16.913  73.689  25.174   73.43
  37.925  73.113  44.289  71.736  45.003  69.622  61.665  71.176  68.414  71.351
    87.4  71.529 110.594  71.043 120.649   69.54 142.133  68.702 157.323  67.651
 187.245  68.626 207.572  69.513 234.933  69.122 238.046   69.71  247.12  69.897
 252.346  69.959 270.002  68.641 277.607  71.686 278.889  72.858 282.069  74.035
 286.421  77.385  287.79  77.395 293.809  77.437 294.876  76.981  302.68  77.437
#Mann= 3 , 0 , 0
       0    .033       0       0    .033       0  302.68    .033       0
Bank Sta=0,302.68
XS Rating Curve= 0 ,0
Exp/Cntr=0.3,0.1

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
Type RM Length L Ch R = 1 ,15006.05,9.944,9.944,9.944
BEGIN DESCRIPTION:
Topo1  9124.758
END DESCRIPTION:
XS GIS Cut Line= 3
992669.039850684176192.383600121992521.270155671 176188.56859896
992373.500460658176184.753597799
#Sta/Elev= 30
       0  75.1381.830994  74.366 2.97998  74.91511.82199  75.138  18.328  69.334
41.96599  66.87449.61099   67.42  53.258  64.83958.43799  64.275  66.297  66.088
  73.842  66.38385.47899  64.462  90.187  64.349  92.355  66.14694.85599  67.208
 105.105  67.586 128.237  66.614 128.567  66.134  142.78  63.786 178.956   65.88
 198.587  64.324 213.736  64.677 214.386  66.162 214.518  67.116 231.291  68.423
 244.751  68.157 254.175   70.44 281.152  71.071 288.546  75.564 295.637  75.884
#Mann= 3 , 0 , 0
       0    .033       0       0    .033       0 295.637    .033       0
Bank Sta=0,295.637
XS Rating Curve= 0 ,0
Exp/Cntr=0.3,0.1

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
Type RM Length L Ch R = 1 ,14638.12,9.978,9.978,9.978
BEGIN DESCRIPTION:
Topo1  9492.683
END DESCRIPTION:
XS GIS Cut Line= 3
992632.175973572175802.265790316992488.795316343175828.555505257
992345.414659114175854.845220199
#Sta/Elev= 29
       0  73.697   4.314  73.697   5.602  73.538  13.911   68.02  18.935  67.887
  26.812  67.528  35.537  66.923  43.765  67.005  52.459  66.668  56.068  66.256
  64.218  66.583  71.209  67.743  75.194  66.888  76.561  65.689  78.424   63.57
 108.893  62.903 132.134  63.396 168.912  65.695 190.325  66.174 207.825  66.409
 212.424  68.585 231.125   68.68 237.799    67.8 260.199  66.791 273.508  67.054
 280.574   72.57 287.488  72.696 289.458  72.043 291.541  72.696
#Mann= 3 , 0 , 0
       0    .033       0       0    .033       0 291.541    .033       0
Bank Sta=0,291.541
XS Rating Curve= 0 ,0
Exp/Cntr=0.3,0.1

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
Type RM Length L Ch R = 1 ,13770   ,9.854,9.854,9.854
BEGIN DESCRIPTION:
Topo1  10360.880
END DESCRIPTION:
XS GIS Cut Line= 3
992278.001436483174964.151311982992153.951880729175047.439850911
992029.902324974 175130.72838984
#Sta/Elev= 30
       0  69.696   4.585  69.696   6.921  69.265  18.676   64.06  32.026  64.188
  36.137  63.172  51.892  63.779  58.878  60.249  65.648  57.467   83.42  57.202
 110.123  58.389 130.887  59.544 134.734  60.288 139.963  60.854 145.303  60.216
 179.105  58.917 203.902  57.762 211.888  60.063 212.807  60.992 231.491  63.622
 240.364  64.241 242.714  65.474 249.516   65.51 257.806  65.218 272.086  65.286
 283.874   64.58 287.928  67.972 295.952  67.848 296.881  67.542 298.832  67.972
#Mann= 3 , 0 , 0
       0    .033       0       0    .033       0 298.832    .033       0
Bank Sta=0,298.832
XS Rating Curve= 0 ,0
Exp/Cntr=0.3,0.1

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
Type RM Length L Ch R = 1 ,13641.9 ,9.709,9.709,9.709
BEGIN DESCRIPTION:
Topo1  10488.943
END DESCRIPTION:
XS GIS Cut Line= 3
992198.729515143174858.542415692992076.849458771174945.274188156
991954.969402398 175032.00596062
#Sta/Elev= 28
       0  68.751   4.454  68.751   6.778  68.077  14.316  63.802  28.104  63.137
  30.364  63.814  46.844  63.577  50.513  58.311  65.317  56.481  86.505  57.009
  97.856  57.033 115.995  60.358 120.137  62.288  129.17  62.912 152.548   63.61
 166.995   63.17 183.098  63.444 195.117  64.011 207.881   63.72 223.445  63.637
 242.153  64.305 256.148   63.61 268.626   62.73 282.812  62.679  288.73  67.383
 296.448   67.38 297.413  66.953 299.179  67.383
#Mann= 3 , 0 , 0
       0    .033       0       0    .033       0 299.179    .033       0
Bank Sta=0,299.179
XS Rating Curve= 0 ,0
Exp/Cntr=0.3,0.1

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
Type RM Length L Ch R = 1 ,13331.2 ,9.947,9.947,9.947
BEGIN DESCRIPTION:
Topo1  10799.605
END DESCRIPTION:
XS GIS Cut Line= 3
992028.478447718174600.895614331991905.717874505174686.005024307
991782.957301292174771.114434284
#Sta/Elev= 29
       0  66.843   3.311  66.936   5.028  66.595  11.587  62.966  26.484  62.186
  37.817  62.967  52.662  63.589  68.881  62.783  78.359  61.801   80.08  60.303
  80.362  58.946  86.337   57.19 106.107  57.152 141.439  57.211 154.159  60.448
 156.285   62.89 168.637   62.57 181.474  62.573 196.384  62.335 210.963   62.49
 225.072   62.45  240.94  62.114 257.343  61.547 270.788  61.959 282.529  62.075
 288.695  66.179 295.171  66.129 296.833  65.849 298.755   65.83
#Mann= 3 , 0 , 0
       0    .033       0       0    .033       0 298.755    .033       0
Bank Sta=0,298.755
XS Rating Curve= 0 ,0
Exp/Cntr=0.3,0.1

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
Type RM Length L Ch R = 1 ,12903.5 ,9.846,9.846,9.846
BEGIN DESCRIPTION:
Topo1  11227.385
END DESCRIPTION:
XS GIS Cut Line= 3
991806.548373794174258.345751511991671.353250727174332.706501454
 991536.15812766174407.067251398
#Sta/Elev= 30
       0  65.036  14.141   65.03   23.12   60.87  33.444  60.146  40.729  61.007
  49.079  63.871  54.039   61.95  63.777  62.407  78.249  62.233  82.351  60.653
  86.587  60.306 105.733  55.197 156.141  59.322 160.011  60.124 176.322  61.231
 179.393  58.196 185.608   58.54  189.02  60.103 190.234  61.717 240.526  61.488
  254.24  61.017 255.438  59.822 259.263  59.874 259.773  61.062 269.899   61.63
 282.448  61.724 295.643  61.159 300.408  62.916 303.466   64.84 308.591  64.761
#Mann= 3 , 0 , 0
       0    .033       0       0    .033       0 308.591    .033       0
Bank Sta=0,308.591
XS Rating Curve= 0 ,0
Exp/Cntr=0.3,0.1

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
Type RM Length L Ch R = 1 ,12647.5 ,9.789,9.789,9.789
BEGIN DESCRIPTION:
Topo1  11483.305
END DESCRIPTION:
XS GIS Cut Line= 3
991652.147140933174038.856130668991535.887028495 174117.11867522
991419.626916057174195.381219773
#Sta/Elev= 30
       0  63.514   6.101   63.79   7.781  63.716  13.522  59.906  17.036  59.422
   51.88  58.128  60.024  58.753  75.592  58.833  79.796  57.519   93.27  57.175
  99.587  55.453 110.499  55.471 111.972  54.875 125.707  53.745 137.452  53.908
 146.013  54.727 147.429  55.366  161.63  55.951 170.544   56.51 176.031  55.248
 183.808  54.954 195.338  53.761 212.519  53.537  222.09  54.001 223.284  55.256
 227.712  56.424  251.17  57.085 267.176  57.847 275.217  64.038 280.295  63.649
#Mann= 3 , 0 , 0
       0    .033       0       0    .033       0 280.295    .033       0
Bank Sta=0,280.295
XS Rating Curve= 0 ,0
Exp/Cntr=0.3,0.1

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
Type RM Length L Ch R = 1 ,12461.5 ,9.5,9.5,9.5
BEGIN DESCRIPTION:
Topo1  11669.316
END DESCRIPTION:
XS GIS Cut Line= 3
991536.569668682173885.793880028 991424.97271301173967.822059584
991313.375757337 174049.85023914
#Sta/Elev= 30
       0  62.584   3.963  62.584   5.483  62.566   8.822  59.373   23.75  58.397
  29.071  58.374  34.852  58.585  40.509  59.433  46.266  57.257  64.799  57.257
  78.353  57.551  94.501  58.215 100.443  55.071 101.977  53.707 110.923  52.391
 124.637  52.976 158.176   54.33 180.808  54.248 200.934  55.071 204.225  56.603
 213.375  56.714 225.345  56.504 237.793  56.667 248.365  56.785 256.584  56.901
 261.414  59.722  262.27  59.813 271.685  60.813 273.463  62.568 277.001  62.568
#Mann= 3 , 0 , 0
       0    .033       0       0    .033       0 277.001    .033       0
Bank Sta=0,277.001
XS Rating Curve= 0 ,0
Exp/Cntr=0.3,0.1

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
Type RM Length L Ch R = 1 ,12347.5 ,9.863,9.863,9.863
BEGIN DESCRIPTION:
Topo1  11783.333
END DESCRIPTION:
XS GIS Cut Line= 3
991473.356639698173794.352036127 991357.39719254 173876.09578881
991241.437745382173957.839541492
#Sta/Elev= 27
       0  61.536    4.52   61.51   6.168  61.212   9.329  58.023  25.575  58.095
  34.919  58.397  38.922  56.793  65.416  56.533  86.743  56.836 101.583  57.259
 106.911  55.276  108.28   53.56 117.997  52.194 142.814   52.66 161.704  53.131
 189.454  53.531 203.165  54.655 205.346  55.254 222.923   55.76 227.741  57.638
  236.53  57.731 248.885  57.213 266.114  56.718 274.912  56.594 280.383   60.67
 281.014  60.679  283.75   60.72
#Mann= 3 , 0 , 0
       0    .033       0       0    .033       0  283.75    .033       0
Bank Sta=0,283.75
XS Rating Curve= 0 ,0
Exp/Cntr=0.3,0.1

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
Type RM Length L Ch R = 1 ,11814.9 ,9.881,9.881,9.881
BEGIN DESCRIPTION:
Topo1  12315.971
END DESCRIPTION:
XS GIS Cut Line= 3
991191.551933657173352.103879808991065.762270016173434.579444517
990939.972606374173517.055009225
#Sta/Elev= 30
       0  58.813   4.834  58.813   9.753  58.651  13.137   56.06  19.078  55.611
  23.902  52.428  39.464  52.169  59.121  52.059  70.966  49.659  74.885  48.014
  90.855  47.408 110.133  47.368 126.827  48.166  141.04   48.95 159.419  48.631
 178.918   49.06 189.107  48.788 203.208  48.903 216.775  47.077 227.416  46.757
 234.531  48.003 237.228  49.667 242.914  50.888 257.584  50.841 266.592  51.574
 275.903   51.27 286.132  51.656 292.794  54.856 296.774  58.583 300.833  58.583
#Mann= 3 , 0 , 0
       0    .033       0       0    .033       0 300.833    .033       0
Bank Sta=0,300.833
XS Rating Curve= 0 ,0
Exp/Cntr=0.3,0.1

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
Type RM Length L Ch R = 1 ,11656.8 ,9.978,9.978,9.978
BEGIN DESCRIPTION:
Topo1  12474.084
END DESCRIPTION:
XS GIS Cut Line= 3
991111.669745379 173223.73142703990980.812204608173301.624409216
990849.954663837173379.517391402
#Sta/Elev= 29
       0  58.122    4.33  58.113   5.919  57.869  15.549  53.073  28.592  52.644
  43.803  52.625  45.859  51.274  66.982  52.339  88.555  51.567  94.193  49.743
 100.087  47.278 114.694  44.926 146.153  45.986 160.988  46.919 178.445  49.885
 184.767  51.902 199.173  50.786 210.803   50.92 220.096  49.764 221.216  49.028
 225.693  49.739   227.4  50.698  233.49  51.657 258.772  51.854  284.23  51.048
 290.705  52.087 296.565  58.061 300.539  58.112 304.571  57.116
#Mann= 3 , 0 , 0
       0    .033       0       0    .033       0 304.571    .033       0
Bank Sta=0,304.571
XS Rating Curve= 0 ,0
Exp/Cntr=0.3,0.1

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
Type RM Length L Ch R = 1 ,10748.8 ,9.759,9.759,9.759
BEGIN DESCRIPTION:
Topo1  13382.052
END DESCRIPTION:
XS GIS Cut Line= 3
990606.692924364172463.539886329 990479.84406152172547.246599969
990352.995198675 172630.95331361
#Sta/Elev= 30
       0  53.588   4.321   53.59   6.689  53.337  16.387  46.217  28.372  46.273
  32.187   46.49  46.288   46.99  61.534  46.518  72.971  45.254  86.266  45.649
  91.011  44.261  99.914  43.638 112.293  43.519 133.681   42.48 148.723  43.122
 163.502  43.877 170.038  43.371 196.358  42.678  212.08  42.389 217.156  44.253
 217.931  44.659 235.645  44.534 249.709  44.707 259.393  45.476 270.195  45.324
 283.872  46.155 293.802  47.086 299.977  53.419 300.814   53.35 303.956  53.419
#Mann= 3 , 0 , 0
       0    .033       0       0    .033       0 303.956    .033       0
Bank Sta=0,303.956
XS Rating Curve= 0 ,0
Exp/Cntr=0.3,0.1

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
Type RM Length L Ch R = 1 ,10465.8 ,9.317,9.317,9.317
BEGIN DESCRIPTION:
Topo1  13665.077
END DESCRIPTION:
XS GIS Cut Line= 3
990467.623050253172237.124046258990332.811885616172305.623771231
990198.000720978172374.123496205
#Sta/Elev= 30
       0  52.316   4.153  52.316   5.871  52.018  18.012  45.489   39.84   47.11
    43.3  47.101  60.585  46.957  63.959  45.746  75.615  46.029  92.184  46.277
 102.635  46.387 116.543   46.13 120.251  44.174 123.151  41.981 128.763  41.147
 156.648  40.323 175.848  40.367 194.518  40.392 215.047  42.176 218.293  44.138
 222.733  46.105  237.84  45.677 253.422  44.501 265.716  46.023 277.638  45.583
 289.343   45.37 293.343   45.87 298.828  51.755 299.502  51.686 302.431  51.755
#Mann= 3 , 0 , 0
       0    .033       0       0    .033       0 302.431    .033       0
Bank Sta=0,302.431
XS Rating Curve= 0 ,0
Exp/Cntr=0.3,0.1

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
Type RM Length L Ch R = 1 ,10354   ,9.993,9.993,9.993
BEGIN DESCRIPTION:
Topo1  13776.881
END DESCRIPTION:
XS GIS Cut Line= 3
990426.898670095172146.887498118990287.209151001172203.759261169
990147.519631907 172260.63102422
#Sta/Elev= 30
       0  51.891   4.371  51.891  14.868  47.939  38.558    48.2  51.658  48.059
  58.814  46.512  70.941  46.071  74.111  47.726  80.596  45.272   96.99  46.363
 109.404  46.805 120.044  46.867 125.781  44.041 127.154  41.877 133.506  40.875
 158.459  39.386 179.184  40.387 205.552    39.4 228.325   42.96 232.165  44.263
 237.113  44.719 243.652  46.504 247.745   46.79 273.876  46.437 288.162  45.508
 292.161  45.508 296.253  48.307 298.249  51.328 298.259  48.328 301.645  51.332
#Mann= 3 , 0 , 0
       0    .033       0       0    .033       0 301.645    .033       0
Bank Sta=0,301.645
XS Rating Curve= 0 ,0
Exp/Cntr=0.3,0.1

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
Type RM Length L Ch R = 1 ,9484.6  ,9.4,9.4,9.4
BEGIN DESCRIPTION:
Topo1  14646.277
END DESCRIPTION:
XS GIS Cut Line= 3
990242.613039699171358.958600109990084.763346112171365.961749725
989926.913652524171372.964899341
#Sta/Elev= 30
       0  47.589   4.202  47.589  13.855  47.218  14.321  43.754  19.628  41.446
  35.636  40.976  50.232  41.312  65.047  41.014  78.178  41.473  86.267  32.694
 112.559  33.465 122.559  33.465 136.528  34.179  144.84  35.673 155.191  36.349
 170.159  36.679  176.22  40.203 183.578  40.819  194.64  40.862 208.509  41.347
 213.471  36.196 225.137   36.06 242.373  36.355 258.147  37.758 258.562  39.958
 267.173  40.197  291.84  40.385 303.521  41.182  310.94  47.332 316.009  47.332
#Mann= 3 , 0 , 0
       0    .033       0       0    .033       0 316.009    .033       0
Bank Sta=0,316.009
XS Rating Curve= 0 ,0
Exp/Cntr=0.3,0.1

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
Type RM Length L Ch R = 1 ,9353    ,9.685,9.685,9.685
BEGIN DESCRIPTION:
Topo1  14777.806
END DESCRIPTION:
XS GIS Cut Line= 3
990233.198480981 171237.34916998990073.433937024171235.660629763
989913.669393066171233.972089547
#Sta/Elev= 30
       0   47.01   4.324   47.01   6.511  46.756  15.151  41.422  31.927  41.011
  56.088  41.182  60.146  39.517  74.476  40.167  79.143  41.286  89.985  41.764
  97.333  33.764 108.299  32.836 125.433  32.866 133.434  33.066 140.916  33.654
   158.4  33.597 165.409  34.812 185.323  36.626 198.343  35.764  211.17  35.922
 226.281  36.048 245.555  36.071 258.121  36.279 263.179  42.109 281.197   40.76
   297.3  39.928 306.819  40.529 313.804   46.43 314.483  46.419 319.546   46.43
#Mann= 3 , 0 , 0
       0    .033       0       0    .033       0 319.546    .033       0
Bank Sta=0,319.546
XS Rating Curve= 0 ,0
Exp/Cntr=0.3,0.1

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
Type RM Length L Ch R = 1 ,9101.2  ,9.779,9.779,9.779
BEGIN DESCRIPTION:
Topo1  15029.633
END DESCRIPTION:
XS GIS Cut Line= 3
990263.809135583171011.718153773990107.754766247170986.396012928
989951.700396912170961.073872084
#Sta/Elev= 30
       0  45.538    6.43  45.302   13.55  40.781  20.816  40.472  32.448  40.236
  45.462  40.657  59.518  39.833  89.831  39.083  93.899  40.183 119.948  40.929
 136.108    31.8 141.029   31.63 152.674  32.266 156.594   33.28 172.615  33.116
 184.727  32.685 190.233  32.083 205.726  31.691 215.726  32.691 216.638  33.765
 243.129  33.676 251.129  35.676 252.107  39.529 261.853  40.287 270.474  40.457
 283.158  39.972 294.042  38.884 300.337  39.519 307.534  45.071  316.19  45.071
#Mann= 3 , 0 , 0
       0    .033       0       0    .033       0  316.19    .033       0
Bank Sta=0,316.19
XS Rating Curve= 0 ,0
Exp/Cntr=0.3,0.1

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
Type RM Length L Ch R = 1 ,8827.4  ,9.809,9.809,9.809
BEGIN DESCRIPTION:
Topo1  15303.406
END DESCRIPTION:
XS GIS Cut Line= 3
990307.256950325170743.749481804990147.993835383170716.425891392
989988.730720441170689.102300979
#Sta/Elev= 30
       0  44.439   4.621  44.286  13.552  44.439  18.909  40.478  30.366  40.268
  50.685  40.133  63.717  39.102   75.85  31.423  77.843  30.676  92.374   30.66
 107.374   30.66 110.816   31.62 126.398   31.72  142.16  31.709 159.321  32.239
 173.927  31.841 194.073  32.366 214.282  32.579 236.937  33.352 256.119  32.061
 257.962  39.735 262.126  39.392 273.062  39.507 290.407  38.646   301.9  39.383
 306.679  43.711 308.187  43.622 310.873  43.464 314.332  41.371 323.179  43.711
#Mann= 3 , 0 , 0
       0    .033       0       0    .033       0 323.179    .033       0
Bank Sta=0,323.179
XS Rating Curve= 0 ,0
Exp/Cntr=0.3,0.1

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
Type RM Length L Ch R = 1 ,8611.6  ,9.824,9.824,9.824
BEGIN DESCRIPTION:
Topo1  15519.276
END DESCRIPTION:
XS GIS Cut Line= 3
990351.754997243170541.819968192990199.062537765 170506.77069486
990046.370078288170471.721421528
#Sta/Elev= 30
       0   43.11   4.901  43.197    7.02  42.897  14.954   38.82  20.695  38.763
  32.369  36.123  37.978  35.591  42.495  33.293  57.976  33.848  78.014   31.27
   93.69   30.61 110.652  30.133 129.052   30.48 140.587   30.96 160.489  30.647
 164.131  29.436  169.03  28.752 185.115  28.594 195.115  28.594 202.617  29.508
 207.368  31.323 235.664   32.39 248.768  32.803 261.662  32.277 292.758  32.476
 298.627  36.996 301.168   37.51 308.081  42.966 310.079  42.828 313.326  42.966
#Mann= 3 , 0 , 0
       0    .033       0       0    .033       0 313.326    .033       0
Bank Sta=0,313.326
XS Rating Curve= 0 ,0
Exp/Cntr=0.3,0.1

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
Type RM Length L Ch R = 1 ,8366    ,9.51,9.51,9.51
BEGIN DESCRIPTION:
Topo1  15764.823
END DESCRIPTION:
XS GIS Cut Line= 3
990396.431169592170279.736823892990241.813103973170265.551024508
990087.195038355170251.365225125
#Sta/Elev= 27
       0  44.194    .225  42.146   3.773  42.138   6.192  41.837  12.538  36.193
  33.911  35.522  40.225  35.578  42.367  32.685  47.818  32.546  52.829  28.474
  66.597  27.721 138.078   29.28 153.631  28.892 158.005  28.277 182.344  28.272
 186.759  28.839 190.829  29.569 206.483  28.531 214.346   28.71 223.836  30.059
  256.91  29.457  273.95  29.463 287.418  28.995 292.572    33.3 298.412  33.694
 306.397   41.45 310.534   41.45
#Mann= 3 , 0 , 0
       0    .033       0       0    .033       0 310.534    .033       0
Bank Sta=0,310.534
XS Rating Curve= 0 ,0
Exp/Cntr=0.3,0.1

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
Type RM Length L Ch R = 1 ,8175.8  ,9.884,9.884,9.884
BEGIN DESCRIPTION:
Topo1  15955.086
END DESCRIPTION:
XS GIS Cut Line= 3
990412.017278141170101.667586265990258.351529529170076.593881883
990104.685780918170051.520177502
#Sta/Elev= 30
       0  41.267    6.55  40.981  12.007  35.012  23.142  34.617  30.265  34.716
  39.757  27.546  51.268  26.671  60.916   26.71  63.337  27.496  77.541  27.711
 103.577  27.857 109.706  27.379 126.164  27.332 129.995  27.917 154.952  28.201
 168.865  27.824 176.403  28.424  188.73  28.516 228.147  28.487  254.52  27.954
 255.264  34.639 266.106  33.707 274.485  34.238 281.812  33.851 296.158  33.677
 298.395  36.735 301.515  37.038 304.901  38.793 307.453  40.692 311.395  40.692
#Mann= 3 , 0 , 0
       0    .033       0       0    .033       0 311.395    .033       0
Bank Sta=0,311.395
XS Rating Curve= 0 ,0
Exp/Cntr=0.3,0.1

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